HEC-RAS study SBPOTOMC.prj: SBPOTOMC

--- SBPOTOMC.g01 (geometry) --- (continued)

Type RM Length L Ch R = 1 ,55391   ,1076.9,771.8,770.2
XS GIS Cut Line= 5
2456839.23266634657501.4117542982458745.09598331656919.745928684
2460456.43658221657437.971911256 2461294.7487957657653.214236342
2462019.77557493658004.399082534
#Sta/Elev= 30
       0 1810.99   639.5 1609.09  798.451572.382   831.7 1553.85  898.691551.411
  998.921537.294  1061.8 1525.96  1116.1  1495.8    1183 1522.83  1222.4 1531.27
 1390.791537.122 1600.331526.652 1700.561517.904  2128.1 1483.99  2157.4 1477.78
 2223.261445.574  2286.9 1425.86  2387.2  1422.2 3765.211420.827  4030.9 1415.21
  4154.7 1423.75  4200.7 1417.48  4282.8 1413.72  4338.7 1417.04    4365 1424.72
  4443.9 1471.34  4476.7 1482.86 4879.981536.917 4891.641538.073  5451.8 1616.59
#Mann= 13 ,-1 , 0
       0      .1       0  798.45     .06       0  898.69    .055       0
  998.92      .1       0 1390.79     .05       0 1600.33      .1       0
 1700.56     .05       0 2223.26     .05       0 3765.21     .05       0
  4200.7    .045       0  4338.7      .1       0 4879.98      .1       0
 4891.64      .1       0
Bank Sta=4200.7,4338.7
XS Rating Curve= 0 ,0
Exp/Cntr(USF)=0,0
Exp/Cntr=0.3,0.1

Type RM Length L Ch R = 1 ,54620   ,1227.8,999.5,1024.6
XS GIS Cut Line= 4
2457432.50806046658780.2682965992459934.70806687658080.352210889
2461142.06331472 658342.820743032461527.01716186658412.812351601
#Sta/Elev= 30
       0 1774.89   340.5 1673.95   462.6 1632.09   538.1 1602.29  712.581521.357
   745.8 1506.23     779  1502.3  812.521485.225   882.9 1469.68   953.5 1429.27
   974.3 1421.42 1212.281417.056  1278.5 1416.88  1294.1 1412.98  1306.5 1416.96
  2721.1  1417.1  2805.5  1420.9  2872.5 1412.32 2932.53 1416.58 2935.371416.527
  3032.2 1417.72  3114.9 1412.96  3175.1    1411  3220.5 1412.64  3309.9 1418.71
  3367.8 1444.85  3477.41451.628 3748.421474.075  4058.1 1528.11  4225.1 1567.82
#Mann= 10 ,-1 , 0
       0      .1       0  712.58     .06       0  812.52     .05       0
 1212.28     .05       0 2932.53     .05       0 2935.37      .1       0
  3114.9    .045       0  3220.5      .1       0  3477.4      .1       0
 3748.42      .1       0
Bank Sta=3114.9,3220.5
XS Rating Curve= 0 ,0
Exp/Cntr(USF)=0,0
Exp/Cntr=0.3,0.1

Type RM Length L Ch R = 1 ,53620   ,759.9,883.5,915.3
XS GIS Cut Line= 4
2458156.74226682659805.6374871962460139.23736629659182.567598791
2460864.26414553659137.2534250892461895.16159725659239.210315919
#Sta/Elev= 30
       0 1665.74   387.8 1571.94  560.361520.999   625.9 1494.34   643.6 1480.42
   677.2 1477.96  761.061425.204   790.4 1411.51   823.9 1408.35  861.411412.696
  935.471412.771  2145.7  1413.5  2173.8 1418.83  2233.9 1409.03 2265.291410.208
    2290 1409.37  2334.1 1406.94  2345.1 1409.82  2382.2 1427.39  2503.6 1429.07
 2564.691437.248  2804.7 1448.79  2847.2 1455.73 3071.341470.797  3160.8 1479.98
 3276.851511.611  3430.1 1558.19 3613.651595.729    3711 1611.08  3840.5 1622.76
#Mann= 12 ,-1 , 0
       0      .1       0  560.36     .06       0  761.06     .05       0
  861.41     .05       0  935.47     .05       0 2265.29      .1       0
    2290    .045       0  2345.1      .1       0 2564.69     .05       0
 3071.34      .1       0 3276.85      .1       0 3613.65      .1       0
#XS Ineff= 1 ,-1
 2435.25 2563.42 1432.18
Permanent Ineff=
       F
Bank Sta=2290,2345.1
XS Rating Curve= 0 ,0
Exp/Cntr(USF)=0,0
Exp/Cntr=0.3,0.1

Type RM Length L Ch R = 1 ,52737   ,682.8,1211.3,829.5
XS GIS Cut Line= 4
2458505.62463119660487.5009044872460098.98876273659934.249469924
 2460311.4373136660075.8818371722461488.75636635659960.805538783
#Sta/Elev= 30
       0 1616.57  122.521587.388   318.8 1546.56     4251513.979   483.9 1492.58
  525.831491.904   581.3 1477.76     636  1468.7   692.8 1449.65   742.2 1439.15
   801.5 1413.13   846.8 1407.47     865 1411.46   983.5 1412.45  1068.2 1409.51
  1271.5 1414.29 1716.061413.456  1787.3 1410.24  1802.3 1405.82  1859.5 1405.46
  1877.3  1409.5 1888.271425.129  1909.1 1433.75  2447.7 1443.88  2753.2 1461.24
  2917.9  1477.5 2997.221497.164  3042.5 1507.56 3096.741514.805  3124.9 1517.09
#Mann= 10 ,-1 , 0
       0     .05       0  122.52      .1       0     425     .06       0
  525.83     .05       0 1716.06      .1       0  1787.3    .045       0
  1877.3      .1       0 1888.27     .05       0 2997.22      .1       0
 3096.74      .1       0
Bank Sta=1787.3,1877.3
XS Rating Curve= 0 ,0
Exp/Cntr(USF)=0,0
Exp/Cntr=0.3,0.1

Type RM Length L Ch R = 1 ,51525   ,461.4,463,463.9
XS GIS Cut Line= 4
2458836.45487235660983.8060034532459289.59660938660904.506199474
2460603.70764674660621.292613836 2461872.5045104660417.378832176
#Sta/Elev= 30
       0 1563.55   72.17 1541.58   128.2 1520.81   229.7  1493.5  270.821486.526
   294.7  1478.8   323.1 1477.87   343.4  1471.4  370.14 1468.25   538.9 1437.73
   579.9 1433.45   616.7 1423.04   645.3 1406.65   682.2 1402.74   735.4 1402.93
   755.8 1406.17  767.821405.665   800.8 1412.03  867.271409.548 1265.061411.847
  1526.1 1426.94  1839.8 1433.78  2062.6 1445.32  2281.4 1472.16  2418.1 1479.33
 2457.551486.264 2556.871509.354 2656.181531.891 2954.131590.175  3089.4 1603.83
#Mann= 13 ,-1 , 0
       0     .05       0   72.17      .1       0  270.82     .06       0
  370.14     .05       0   645.3    .045       0   755.8     .05       0
  767.82      .1       0  867.27     .05       0 1265.06     .05       0
 2457.55      .1       0 2556.87     .12       0 2656.18      .1       0
 2954.13     .12       0
Bank Sta=645.3,755.8
XS Rating Curve= 0 ,0
Exp/Cntr(USF)=0,0
Exp/Cntr=0.3,0.1

Type RM Length L Ch R = 1 ,51062   ,554.7,640.3,917
XS GIS Cut Line= 4
2458604.40772794661429.2922262272459479.41272295661335.205667624
2460761.34208392 661064.70681164 2461771.3496749660866.573296408
#Sta/Elev= 30
       0 1628.83   207.5 1573.45   267.9 1566.06   328.2 1543.45   448.9 1510.29
  571.971482.627     642 1472.35   658.1 1465.37   698.1 1463.84  770.891448.327
   879.7 1435.11   936.6 1423.58   974.3 1405.48  1091.9 1402.62  1100.1  1406.2
  1145.1 1412.04 1268.051409.559 1665.761411.536  1782.8  1413.5  1831.9 1420.38
  2224.2 1439.59  2387.2 1441.25 2461.011447.839 2560.381475.055  2664.5  1499.7
 2858.491527.962 2907.771535.735 2957.861544.353 3057.231557.932  3219.5 1587.12
#Mann= 13 ,-1 , 0
       0     .05       0  571.97     .06       0  770.89     .05       0
   974.3    .045       0  1100.1      .1       0 1268.05     .05       0
 1665.76     .05       0 2461.01     .12       0 2560.38      .1       0
 2858.49      .1       0 2907.77     .12       0 2957.86      .1       0
 3057.23     .12       0
Bank Sta=974.3,1100.1
XS Rating Curve= 0 ,0
Exp/Cntr(USF)=0,0
Exp/Cntr=0.5,0.3

Type RM Length L Ch R = 1 ,50422   ,164,155.1,145.5
XS GIS Cut Line= 5
2458721.28063192661818.3055934282459395.57130594661758.101068961
2460039.75971773662095.2464059722461020.41839018 662116.04941746
2461060.10519367662508.704964611
#Sta/Elev= 30
       01602.644 214.314 1552.88 423.1411496.698   463.3 1487.65  618.941462.862
 680.5551447.028  777.711440.364 788.9081436.964  852.831436.238 883.7171433.298
 906.2911420.991   942.41406.454 969.4961401.5581059.2561401.2281100.4231401.535
    11231405.859 1142.011408.717 1225.091407.797 1306.161406.512 1349.181407.231
  1629.81408.122 1763.321407.6251895.1491409.594 2189.05 1424.21 2268.231424.608
 2369.211424.052 2448.391427.0412484.2781423.786 2546.071424.9782779.5891436.733
#Mann= 16 ,-1 , 0
       0     .05       0  618.94     .06       0  852.83      .1       0
   942.4    .045       0    1123      .1       0 1142.01     .06       0
 1225.09      .1       0 1306.16     .06       0 1349.18     .05       0
  1629.8     .06       0 1763.32     .05       0 2189.05     .06       0
 2268.23    .055       0 2369.21     .05       0 2448.39     .06       0
 2546.07     .05       0
#XS Ineff= 3 ,-1
       0     849    1435    1216 2060.75 1418.17 2285.05 2565.42 1426.82
Permanent Ineff=
       F       F       F
Bank Sta=942.4,1123
XS Rating Curve= 0 ,0
Exp/Cntr(USF)=0,0
Exp/Cntr=0.5,0.3

Type RM Length L Ch R = 1 ,50267   ,132.1,79.4,35.9
XS GIS Cut Line= 5
2458752.99373075662006.0479322752459424.61250147  661943.8184245
2460086.95631354662243.6963725062460907.34299476662251.739891965
2460953.16811935662467.087688934
#Sta/Elev= 30
       0 1589.75  66.0331578.742 258.8551535.381 415.5241490.913 604.3291461.527
 676.8371442.622  725.491438.617 804.1721437.481  835.891429.228  844.681428.229
 899.0671420.313 941.3821404.678 953.4621401.2811023.7151401.1331085.1881401.365
1093.969 1405.381093.9691405.3811168.6141405.492 1192.271413.691 1202.261417.502
1298.0311413.8541331.7221406.406 1370.461407.871 1636.16 1406.921833.3721407.718
1909.3751415.445  1938.51422.995 2140.051427.304 2225.21  1426.52442.1581440.246
#Mann= 12 ,-1 , 0
       0     .05       0  725.49     .06       0  835.89     .05       0
  844.68    .055       0 941.382    .045       01093.969     .06       0
 1192.27      .1       0 1202.26     .06       0 1370.46     .05       0
 1636.16     .06       0  1938.5      .1       0 2140.05     .05       0
#XS Ineff= 1 ,-1
 1209.44 1944.44 1418.46
Permanent Ineff=
       F
Bank Sta=941.382,1093.969
XS Rating Curve= 0 ,0
Exp/Cntr(USF)=0,0
Exp/Cntr=0.5,0.3

Type RM Length L Ch R = 1 ,50188   ,87,85.3,38.5
XS GIS Cut Line= 6
2458765.47016644662259.8110958782459634.50029789662165.972161496
 2459901.7372632662170.0521151642460109.81490031662261.851072713
2460839.49775751662359.1615176152460925.89060745662512.073470475
#Sta/Elev= 30
       01569.341 226.5841532.035 407.6311486.053 447.8631484.251 504.1891470.266
 620.8631455.992 689.258 1440.04 781.7931429.843  801.911423.276  844.211421.636
  906.751416.797 930.3331403.962 970.3381401.111    10581403.885 1062.061404.507
1110.3541405.7951126.3561417.595 1147.291417.7461212.797 1414.581262.3461405.957
 1297.43 1407.49 1797.241407.7111809.5761414.3841841.8591417.2971858.0011430.692
1874.143  1428.4 1900.991439.2311954.851 1444.48 2114.77 1437.29 2280.551446.232
#Mann= 10 ,-1 , 0
       0     .05       0  844.21    .055       0 930.333    .045       0
    1058     .06       0 1062.06      .1       0 1147.29     .06       0
 1297.43     .05       0 1797.24     .06       0 1900.99      .1       0
 2114.77     .05       0
#XS Ineff= 2 ,-1
  -57.08  864.911419.974 1148.39 1993.571420.127
Permanent Ineff=
       F       F
Bank Sta=930.333,1058
XS Rating Curve= 0 ,0
Exp/Cntr(USF)=0,0
Exp/Cntr=0.5,0.3

Type RM Length L Ch R = 1 ,50102   ,300.9,305.5,234.2
XS GIS Cut Line= 6
2458758.70911313662327.8880626352459629.77922142662252.408919762
2460001.05500528662252.4089197622460129.57354585662303.408340622
2460771.65252026662387.4303664712460909.53166971662584.578665008
#Sta/Elev= 30
       01566.583 132.5311547.871 240.9351527.591 433.6551481.757 465.7751480.227
  485.851473.726 634.404 1454.34 714.7041436.566  862.971421.174   899.31421.097
   943.31405.474   955.31401.129   999.31400.961  1063.31401.659  1079.31406.096
 1164.691406.0541385.0591408.2451707.7871406.281  1785.11408.7071796.5381415.053
1824.7761416.3541853.0151438.2291865.1171435.641 1877.221442.751 1902.281448.273
1945.7991452.8462031.4311446.044 2063.141448.1692217.0941456.954 2272.011452.251
#Mann= 8 ,-1 , 0
       0     .05       0  862.97     .06       0   943.3    .045       0
  1079.3      .1       0 1164.69     .06       0  1785.1     .06       0
 1902.28      .1       0 2063.14     .05       0
#XS Ineff= 2 , 0
                         1118.04         1419.68
Permanent Ineff=
       F       F
Bank Sta=943.3,1079.3
XS Rating Curve= 0 ,0
Exp/Cntr(USF)=0,0
Exp/Cntr=0.5,0.3

Type RM Length L Ch R = 1 ,49797   ,201.1,580.3,1004.4
XS GIS Cut Line= 4
 2458922.3217186662463.5317454282459473.87101086662549.160402674
2460723.04201069662556.7158724312460889.18416278662781.275324612
#Sta/Elev= 30
       01531.742  12.5721531.799  81.3871518.916 154.2491500.216 364.218 1466.48
 514.5141450.773 554.9931442.504  650.181430.528 759.0341418.418 783.0351403.162
 831.1151403.778 907.0371400.028 959.0381400.151  971.811404.089 991.0391406.608
 1053.031405.443 1556.591405.5451579.0491406.351 1595.051413.558 1623.051415.855
1647.0511437.958  1657.31443.9891687.0511459.5371699.0521460.9151739.0521476.511
1771.0531481.9191853.9281476.994 1917.861467.7741988.434 1469.532086.6891462.812
#Mann= 8 ,-1 , 0
       0     .05       0  650.18     .06       0 831.115    .045       0
  971.81      .1       0 1053.03     .05       0 1556.59     .06       0
  1657.3      .1       0 1917.86     .05       0
#XS Ineff= 1 ,-1
 1293.72 1654.211435.848
Permanent Ineff=
       F
Bank Sta=831.115,971.81
XS Rating Curve= 0 ,0
Exp/Cntr(USF)=0,0
Exp/Cntr=0.5,0.3

Type RM Length L Ch R = 1 ,49216   ,112,90.7,148.9
XS GIS Cut Line= 4
2458930.70829003662496.4484086692459689.57967242662755.525466638
2460048.61559528663667.3951116162460103.69496981663846.913073044
#Sta/Elev= 30
       0 1531.79    16.9 1525.87      55 1519.92     148  1498.3     241 1483.21
   397.3 1462.61   511.5 1453.62   581.7 1440.17  700.84 1422.79   739.3  1422.1
   765.1 1415.05   790.4 1415.57   805.1 1409.12   837.8 1403.75  1102.1 1399.51
    1158 1397.77  1248.3 1399.07  1274.2  1405.6 1316.481405.498  1368.6 1402.47
  1409.9 1407.87 1428.221418.293  1467.5 1420.47  1476.1 1419.31  1484.7 1414.42
 1528.19 1416.06  1656.7 1420.41  1725.5 1426.17  1806.5 1438.06  1969.7 1450.32
#Mann= 7 ,-1 , 0
       0     .05       0  700.84     .06       0  1102.1    .045       0
  1248.3     .06       0 1316.48     .05       0 1428.22     .06       0
 1528.19     .05       0
#XS Ineff= 2 , 0
            1070    1401    1278            1401
Permanent Ineff=
       F       F
Bank Sta=1102.1,1248.3
XS Rating Curve= 0 ,0
Exp/Cntr(USF)=0,0
Exp/Cntr=0.5,0.3

Type RM Length L Ch R = 1 ,49126   ,274.8,275.4,307.9
XS GIS Cut Line= 4
2458900.10863751 662510.728246512459624.30041372662786.125119154
2459887.45742536663579.6761077372459977.21640607663873.432771891
#Sta/Elev= 30
       0 1532.53    23.9 1531.65    41.3 1525.86   183.8  1496.3   268.1 1483.62
     465 1458.63   542.9 1453.73     679 1430.24  751.891422.796   780.5 1420.38
   796.3 1414.88     828 1414.69     843 1410.16   851.5 1411.58   864.1 1406.47
  879.441405.964  1070.6 1400.09  1081.1 1397.17  1154.9 1397.49  1171.7 1400.47
  1218.1 1414.31 1275.341418.531  1340.6 1420.59  1390.9 1427.96  1424.6 1424.74
 1472.83 1424.88  1760.6 1432.93    1815 1433.01  1844.2 1429.49    1918 1437.53
#Mann= 7 ,-1 , 0
       0     .05       0  751.89     .06       0  879.44    .025       0
  1070.6    .045       0  1171.7     .05       0 1275.34     .06       0
 1472.83     .05       0
Bank Sta=1070.6,1171.7
XS Rating Curve= 0 ,0
Exp/Cntr(USF)=0,0
Exp/Cntr=0.5,0.3

Type RM Length L Ch R = 1 ,48850   ,310.4,305.3,302.1
XS GIS Cut Line= 4
2458898.06866067662539.2879221912459416.22277661662953.403219575
2459520.26159517663334.878887609 2459646.7401589663773.473907005
#Sta/Elev= 30
       0 1531.22    79.9 1520.02   144.2 1506.64   304.7 1482.15  490.011459.493
   555.2 1453.47  622.381440.966   685.6 1430.34   714.6 1429.38   718.7 1425.57
     727  1406.6  731.12 1402.47     748 1398.94   775.8 1397.91   803.4 1395.41
   834.8 1395.22   863.9 1395.56   881.6 1398.31   921.9 1411.26   930.2 1418.59
   938.5 1422.64   988.2 1429.45  1004.8  1441.3 1025.581449.061  1057.5  1456.3
  1096.2 1458.89 1123.851458.824  1183.6 1460.17  1341.8 1459.63  1515.2 1468.07
#Mann= 8 ,-1 , 0
       0     .05       0  490.01      .1       0  622.38     .06       0
  731.12      .1       0   775.8    .045       0   881.6     .05       0
 1025.58      .1       0 1123.85     .05       0
Bank Sta=775.8,881.6
XS Rating Curve= 0 ,0
Exp/Cntr(USF)=0,0
Exp/Cntr=0.3,0.1

Type RM Length L Ch R = 1 ,48545   ,677.4,673.2,667.7
XS GIS Cut Line= 4
2458817.60787106662552.8007919152459082.50777871662950.150653391
2459257.10089966663353.5209673152459395.57130594663811.075353258
#Sta/Elev= 30
       0 1540.41    69.8 1530.61   137.1 1524.13   276.3 1500.77  396.821484.853
  502.641470.983   520.9 1464.44   530.7 1458.35     535  1453.8   543.7 1435.86
   548.1 1429.09   565.5 1413.64   569.9 1411.76     596 1410.47  603.431407.706
   612.1 1399.77   617.8 1396.09   636.5 1395.38   691.9 1395.74   703.4 1399.42
  704.211399.855   748.6 1410.71   774.7 1427.24     814 1438.46   948.4 1487.31
     977 1492.95 1004.521493.454  1165.1  1492.9  1307.7 1502.99  1395.1 1505.32
#Mann= 8 ,-1 , 0
       0     .05       0  396.82      .1       0  502.64     .06       0
  603.43      .1       0   612.1    .045       0   703.4      .1       0
  704.21      .1       0 1004.52     .05       0
Bank Sta=612.1,703.4
XS Rating Curve= 0 ,0
Exp/Cntr(USF)=0,0
Exp/Cntr=0.3,0.1

Type RM Length L Ch R = 1 ,47872   ,372.3,361.7,356
XS GIS Cut Line= 4
2458161.37855438662625.0462212742458420.25800959 663130.76422679
2458661.07610745663630.4617798592458841.68968085663997.709379103
#Sta/Elev= 30
       0 1536.17  101.911541.057  307.351548.348  410.071550.878   563.8 1552.76
   638.4 1544.41     651  1538.8   657.1 1530.25   680.9  1457.4   683.7 1449.88
   723.7 1426.56   741.4 1407.77   763.6 1406.41   773.8 1399.59   785.8 1394.94
   868.7 1394.04   914.6 1398.44   932.4 1403.23   971.6 1429.27   974.6 1441.93
   981.2  1494.1   985.7 1516.37  1001.6 1543.79 1022.91 1548.95 1030.131551.439
  1056.7 1550.88 1124.861566.527 1227.051581.172 1372.65 1592.77  1532.1 1605.14
#Mann= 12 ,-1 , 0
       0     .05       0  101.91     .06       0  307.35      .1       0
  410.07      .1       0   680.9      .1       0   773.8    .045       0
   914.6      .1       0 1022.91     .12       0 1030.13      .1       0
 1124.86     .12       0 1227.05      .1       0 1372.65     .05       0
Bank Sta=773.8,914.6
XS Rating Curve= 0 ,0
Exp/Cntr(USF)=0,0
Exp/Cntr=0.3,0.1

Type RM Length L Ch R = 1 ,47510   ,873.6,846.5,739.7
XS GIS Cut Line= 4
2458016.62439775662895.2992129392458137.03344672663390.314192006
2458397.91971947663871.9503878552458685.56355866664166.283618651
#Sta/Elev= 30
       0 1551.94   47.171551.396  145.061546.226  242.951531.082   304.2 1522.48
   378.9 1508.73   532.9 1463.27     551 1456.87   576.1 1442.57   587.9 1432.68
   601.1 1411.55   605.6 1406.68   632.1 1407.29  641.721404.518   649.8 1398.77
   660.2 1393.05   705.9 1392.66   755.8 1393.09   764.9 1398.74   778.5 1402.53
   828.5 1434.85  848.821445.997   882.6 1461.65  952.361471.904   978.61475.231
  1028.7 1484.24  1081.3 1500.52 1175.531523.486 1184.791525.431  1468.8 1580.35
#Mann= 12 ,-1 , 0
       0      .1       0   47.17     .06       0  145.06      .1       0
  242.95      .1       0  641.72    .025       0   649.8    .045       0
   764.9      .1       0  848.82     .12       0  952.36      .1       0
   978.6      .1       0 1175.53      .1       0 1184.79      .1       0
Bank Sta=649.8,764.9
XS Rating Curve= 0 ,0
Exp/Cntr(USF)=0,0
Exp/Cntr=0.3,0.1

Type RM Length L Ch R = 1 ,46664   ,758.1,765.8,745.9
XS GIS Cut Line= 4
2457378.71973632  663558.21635052457577.39466706663889.341235064
 2457764.0286929664214.4456671812457974.74452854664569.652361532
#Sta/Elev= 30
       0  1551.7   81.051547.657   147.8 1545.28   300.8 1529.07     362 1514.48
   379.5  1504.9   397.1 1499.17   408.8 1487.16   434.1 1485.39   457.1 1471.61
   461.2  1456.9   466.3 1424.51   470.3 1413.11   477.2 1405.15   499.6 1390.26
   543.6 1387.43   623.2 1387.61  633.56 1390.14   660.1 1403.69   664.7 1421.17
   669.3 1456.04   673.9  1476.3   683.1 1487.91   701.8 1500.02   747.7 1516.34
   840.6 1535.79   887.1 1548.58  920.241551.677  921.53 1551.76    1174  1553.3
#Mann= 6 ,-1 , 0
       0     .05       0   81.05      .1       0   499.6    .045       0
  633.56      .1       0  920.24      .1       0  921.53      .1       0
Bank Sta=499.6,633.56
XS Rating Curve= 0 ,0
Exp/Cntr(USF)=0,0
Exp/Cntr=0.3,0.1

Type RM Length L Ch R = 1 ,45898   ,461.8,429.6,422.2
XS GIS Cut Line= 4
2456772.28558183664130.8938281272456943.45306534664310.839131304
2457228.73220452664714.6188359942457417.45532736664947.231057174
#Sta/Elev= 30
       0 1516.69    32.6 1512.25      50 1503.84    55.8 1502.53    84.8 1503.03
   104.9 1495.47   142.9 1486.46   177.7 1475.77   236.6 1460.12   297.4  1441.1
   339.7  1421.6     377 1408.53     410 1392.12   424.7 1388.09   439.4 1381.86
   448.2 1380.28   496.7 1379.04     555 1380.25   568.6 1381.79   589.4 1385.31
   600.9 1391.09   610.8 1397.69   638.2 1409.47     663  1421.9   679.4 1428.06
   728.4 1442.86   775.6 1454.23   835.8 1473.51   949.1 1489.62  1042.3 1497.55
#Mann= 3 ,-1 , 0
       0      .1       0   439.4    .045       0   568.6      .1       0
Bank Sta=439.4,568.6
XS Rating Curve= 0 ,0
Exp/Cntr(USF)=0,0
Exp/Cntr=0.3,0.1

Type RM Length L Ch R = 1 ,45468   ,521.4,457.2,404.3
XS GIS Cut Line= 4
2456539.67336065664604.8960901542456684.50738515664732.174475328
  2456952.230885664995.5090653432457167.28746685665153.509819352
#Sta/Elev= 30
       0 1569.32   60.871544.235   105.3 1529.17   119.8 1514.08   124.2 1511.34
   154.5 1512.68   165.1 1510.57   201.6  1484.7  218.891467.009   230.9 1457.08
   253.7 1419.57   274.5 1406.33     301 1384.86   315.1 1376.82   347.4 1375.02
   405.6 1377.15     426 1381.31  432.151386.552   437.2 1400.61   442.8 1412.22
     482 1431.15   527.3 1457.67   532.6 1462.76   538.9 1473.71   543.8 1479.18
  554.691486.672   571.5 1495.49   645.9 1514.48   784.9 1533.53   835.2 1535.88
#Mann= 7 ,-1 , 0
       0     .06       0   60.87      .1       0  218.89      .1       0
   315.1    .045       0   405.6      .1       0  432.15      .1       0
  554.69      .1       0
Bank Sta=315.1,405.6
XS Rating Curve= 0 ,0
Exp/Cntr(USF)=0,0
Exp/Cntr=0.3,0.1

Type RM Length L Ch R = 1 ,45011   ,444.9,423.7,395.4
XS GIS Cut Line= 4
2456329.00568863665329.0662126952456596.72918848 665298.34384386
2456908.34178667665276.3992946922457114.62054885665250.065835691
#Sta/Elev= 30
       0 1674.39    13.8 1657.45    62.1 1617.18   114.5 1578.25   138.6 1554.62
   164.11534.833   203.1 1498.89   235.3 1496.46  263.521474.389   295.6 1449.14
   315.6 1414.75   339.7 1390.86   349.5 1375.61   359.7 1371.68   411.8 1371.14
   439.9 1374.42     468 1380.46   500.1 1407.86   524.1 1416.17   528.1 1422.85
   532.1 1434.22   536.2 1439.17   552.2 1446.59  562.671456.461   580.3 1469.33
   620.6 1492.14   667.6 1515.37   710.5 1531.14  761.481539.972   789.8 1541.85
#Mann= 7 ,-1 , 0
       0      .1       0   164.1     .06       0  263.52      .1       0
   349.5    .045       0   439.9      .1       0  562.67      .1       0
  761.48      .1       0
Bank Sta=349.5,439.9
XS Rating Curve= 0 ,0
Exp/Cntr(USF)=0,0
Exp/Cntr=0.3,0.1

Type RM Length L Ch R = 1 ,44587   ,486.5,494.6,490.2
XS GIS Cut Line= 4
2456522.11772131665820.6241140572456781.06340149665732.845917385
2457119.00945868665570.4562535432457277.01021269665526.567155207
#Sta/Elev= 30
       0 1703.56    34.5 1677.99    51.3 1660.89    72.5  1643.1  153.391585.714
   204.8 1551.16   220.3 1535.93   241.4 1533.78  254.091523.438   312.1  1480.4
   315.2 1475.67   337.4 1415.47   341.9 1405.16   355.2 1394.33   372.9 1371.69
   384.1 1368.71   412.9 1368.29     475 1372.35   483.9 1376.51   514.9 1401.26
   545.9 1422.85   568.2 1433.73   572.6 1438.97   578.9 1457.03   585.9 1470.31
   599.9 1477.23     617 1491.83   714.5 1538.14   776.8 1562.91   812.3 1566.48
#Mann= 6 ,-1 , 0
       0      .1       0  153.39     .06       0  254.09      .1       0
   372.9    .045       0     475      .1       0   812.3      .1       0
Bank Sta=372.9,475
XS Rating Curve= 0 ,0
Exp/Cntr(USF)=0,0
Exp/Cntr=0.3,0.1

Type RM Length L Ch R = 1 ,44093   ,543.8,549.8,554.3
XS GIS Cut Line= 4
2456776.67449166666272.6818269162457057.56472101666136.625622075
2457347.23277002  665996.18050742457575.45608137665890.846671394
#Sta/Elev= 30
       0 1690.74   74.791636.172   140.1 1595.01  178.451577.313   188.5 1573.27
   200.5  1562.6     229 1560.59   287.3 1520.96   317.9 1503.52   322.3 1498.64
   326.8 1488.62   361.9 1394.08   366.8 1384.61   397.2 1370.25   407.1 1368.32
   504.6 1368.68   511.9 1370.44   541.8 1384.33   580.1 1408.43  593.96 1420.88
   633.5 1449.85   655.5 1469.77   668.7 1477.03  696.421497.796   783.3 1563.08
  799.511577.433   822.9 1597.87   848.6 1614.45   860.7 1618.48   885.4 1619.41
#Mann= 8 ,-1 , 0
       0      .1       0   74.79     .06       0  178.45      .1       0
   397.2    .045       0   511.9      .1       0  593.96     .12       0
  696.42      .1       0  799.51     .12       0
Bank Sta=397.2,511.9
XS Rating Curve= 0 ,0
Exp/Cntr(USF)=0,0
Exp/Cntr=0.3,0.1

Type RM Length L Ch R = 1 ,43543   ,500.8,538.9,564.2
XS GIS Cut Line= 4
 2456939.0641555666759.8508184442457224.34329468666650.128072604
2457575.45608137666505.2940480962457930.95777789666320.959835086
#Sta/Elev= 30
       0 1714.46   90.57 1641.29   188.2  1570.7   205.4 1547.74   231.1 1543.91
   252.5 1529.68  293.511485.638   308.3 1470.95   325.3 1442.76   351.5 1414.78
   386.1 1388.05   407.8 1378.74   471.5 1369.91   493.8 1367.82   576.4 1369.86
   698.2 1427.59   743.1 1458.52   774.8 1487.44   801.8 1500.83   819.8 1522.24
   842.4 1530.28   869.4 1554.87   900.4 1574.61   912.1 1591.04   938.9 1604.15
   950.8 1615.98  1000.1 1638.78 1015.531662.963  1027.1 1673.56  1085.9 1661.97
#Mann= 7 ,-1 , 0
       0      .1       0   90.57     .06       0  293.51      .1       0
   471.5    .045       0   576.4      .1       0   912.1     .12       0
 1015.53      .1       0
Bank Sta=471.5,576.4
XS Rating Curve= 0 ,0
Exp/Cntr(USF)=0,0
Exp/Cntr=0.3,0.1

Type RM Length L Ch R = 1 ,43004   ,577.9,594.9,644.6
XS GIS Cut Line= 4
2457004.89780301667110.9636051312457338.45495036667102.185785464
2457790.51266322667071.4634166282458229.40364658 667036.35213796
#Sta/Elev= 30
       0 1710.54    85.9 1642.89   101.9 1624.86   130.5 1599.45   145.9  1591.1
   180.81562.377   193.9 1552.62   217.9 1528.46   241.9 1525.18  281.021492.358
     310 1472.88     337 1448.74   427.1 1387.18   454.2 1373.17   476.7 1370.04
   622.6 1367.69   634.7 1371.33   650.7 1382.49  680.251392.758   742.5 1423.43
   903.4 1528.19   954.7 1565.28  1011.7 1613.14    1088  1670.5    1131 1696.87
  1152.2 1713.33  1196.3 1735.43  1204.3 1742.05  1216.4 1743.58  1227.1 1740.81
#Mann= 6 ,-1 , 0
       0      .1       0   180.8     .06       0  281.02      .1       0
   476.7    .045       0   634.7    .025       0  680.25      .1       0
Bank Sta=476.7,634.7
XS Rating Curve= 0 ,0
Exp/Cntr(USF)=0,0
Exp/Cntr=0.3,0.1

Type RM Length L Ch R = 1 ,42409   ,517.5,528.4,557.7
BEGIN DESCRIPTION:
Mannings N in channel placed 0.1 because of island in the channel
END DESCRIPTION:
XS GIS Cut Line= 4
2457009.28671284667541.0767688222457364.78840936667650.799514662
2457812.45721238667751.7444408342458312.79293341667808.800268671
#Sta/Elev= 30
       0 1703.51   135.5 1596.41   152.2 1580.53  161.111576.037   223.2  1531.1
   240.1 1512.92   261.1  1509.6  271.951502.175     349 1444.42   443.8 1384.52
  459.711368.423   460.8 1367.61   468.4 1365.41   525.8 1366.76   603.7 1365.98
   644.7 1363.12     657 1363.38   669.3 1367.52   689.8 1384.46  703.581403.363
   730.8 1427.02   812.1  1482.4   861.2 1519.07     989 1619.46 1224.051780.223
    1252 1798.82  1272.1 1807.54  1287.6 1821.23 1327.221831.266  1334.5 1833.85
#Mann= 11 ,-1 , 0
       0      .1       0  161.11     .06       0  271.95      .1       0
  459.71    .025       0   460.8    .045       0   525.8      .1       0
   603.7    .045       0   669.3      .1       0  703.58      .1       0
 1224.05      .1       0 1327.22      .1       0
Bank Sta=460.8,669.3
XS Rating Curve= 0 ,0
Exp/Cntr(USF)=0,0
Exp/Cntr=0.3,0.1

Type RM Length L Ch R = 1 ,41881   ,416.6,480.6,534.3
XS GIS Cut Line= 4
2457000.50889317668032.6346701832457263.84348319668137.968506189
2457610.56736004668304.7470798662457851.95740089668585.637309215
#Sta/Elev= 30
       0 1534.16    6.661533.088    71.2 1515.17    83.5 1510.26    95.8 1501.83
   118.7 1500.96   135.8 1491.35   198.11464.688   269.5 1432.69   316.5 1414.14
   322.7 1409.38   334.4 1392.58   341.1 1385.71     349 1381.03   366.7    1376
   375.6 1369.09   382.4 1365.95   393.4 1362.17   405.7 1361.88   504.3 1362.07
   514.3 1365.99   566.5 1378.56   606.4 1398.93   637.5 1417.56   664.1 1435.44
   754.6 1490.01   828.9 1538.13   895.7 1584.11   987.6 1654.53  1038.7 1689.09
#Mann= 5 ,-1 , 0
       0      .1       0    6.66     .06       0   198.1      .1       0
   382.4    .045       0   514.3      .1       0
Bank Sta=382.4,514.3
XS Rating Curve= 0 ,0
Exp/Cntr(USF)=0,0
Exp/Cntr=0.3,0.1

Type RM Length L Ch R = 1 ,41400   ,619.4,697.1,728
XS GIS Cut Line= 4
  2456899.563967668159.9130553572457053.17581117668436.414374873
2457298.95476186668809.471710728 2457579.8449912669318.585251423
#Sta/Elev= 30
       0 1495.54    12.6 1495.16    30.9  1488.4   93.991472.611     127 1466.03
   168.1 1452.57   236.8 1437.06   303.1 1416.75   333.7 1405.75   368.3 1386.23
   394.3 1373.02   443.4 1367.88   452.1 1365.95   463.6 1362.12   486.9 1361.56
     610 1361.94   628.2  1366.4   654.2 1372.65     690 1383.74   711.8 1394.01
   740.9 1410.58   796.6 1446.35   812.3 1454.91   852.3 1482.08   970.2 1558.04
  1198.7 1697.38  1209.7 1705.55  1226.2 1715.12  1299.8 1762.53  1344.5 1792.89
#Mann= 4 ,-1 , 0
       0     .06       0   93.99      .1       0   452.1    .045       0
   628.2      .1       0
Bank Sta=452.1,628.2
XS Rating Curve= 0 ,0
Exp/Cntr(USF)=0,0
Exp/Cntr=0.3,0.1

Type RM Length L Ch R = 1 ,40703   ,748.2,790.5,819.5
XS GIS Cut Line= 4
2456451.89516397668295.9692601982456522.11772131668651.470956719
2456653.78501632669239.5848744192456732.78539332669656.531308609
#Sta/Elev= 30
       0 1526.68   110.5 1499.33   125.3  1497.4   206.8 1478.25  217.721473.861
   239.5 1472.42   247.6 1468.84   292.5 1457.98  315.341450.139   372.5 1424.43
   394.6 1412.43   442.8 1383.25   469.6 1370.42   492.9 1365.31   529.8 1364.97
   546.2 1360.53   566.7  1360.9   566.7 1360.91   591.3 1359.57   606.9 1361.53
   665.1 1360.45   731.4 1360.97   747.1 1362.61   775.8 1362.68   874.2  1391.4
   925.1 1412.43  1021.3 1460.61  1188.3 1552.43  1261.5 1596.37  1389.4 1675.69
#Mann= 5 ,-1 , 0
       0      .1       0  217.72     .06       0  315.34      .1       0
   566.7    .045       0   747.1      .1       0
Bank Sta=566.7,747.1
XS Rating Curve= 0 ,0
Exp/Cntr(USF)=0,0
Exp/Cntr=0.3,0.1

Type RM Length L Ch R = 1 ,39912   ,713.7,788.2,830
XS GIS Cut Line= 4
2455793.55868894668414.469825705 2455815.5032381668761.193702558
 2455802.3365086669305.4185219232455819.89214794669801.365333118
#Sta/Elev= 30
       0 1485.57  104.381461.191   184.8 1444.46   196.8 1438.63   216.9 1438.45
  300.271416.084  398.81 1387.88   449.1 1369.42  497.921365.163   512.4  1364.8
   528.8 1361.86   585.2 1358.85   601.2 1356.21   713.3 1355.81   749.2 1356.23
   757.2 1358.52   769.2 1362.22   789.2 1363.45   809.2 1369.16   821.3 1374.77
   857.3 1393.81   934.4 1441.07  1009.1 1488.94  1085.4 1539.86  1133.4 1575.97
  1173.5 1602.74  1197.5 1622.01  1249.3 1657.41  1277.5 1678.27  1388.1  1752.1
#Mann= 7 ,-1 , 0
       0     .05       0  104.38     .06       0  300.27      .1       0
  398.81    .055       0  497.92      .1       0   585.2    .045       0
   757.2      .1       0
Bank Sta=585.2,757.2
XS Rating Curve= 0 ,0
Exp/Cntr(USF)=0,0
Exp/Cntr=0.3,0.1

Type RM Length L Ch R = 1 ,39124   ,866.2,821.4,790.2
XS GIS Cut Line= 4
2455297.61187774668265.246891363 2455187.8891319668611.970768216
2455021.11055823 668971.861374572455034.27728773669226.418144918
#Sta/Elev= 30
       0 1567.37   185.3 1496.11     266 1459.62   333.2 1422.21  365.781407.492
   390.8  1392.8     411 1391.38   463.9 1365.99  483.011364.296   494.7 1358.57
   516.8 1354.98     530 1351.81   609.4 1351.47   652.9 1355.02   675.5  1366.1
   693.1 1392.73   715.2 1414.07   719.6 1421.25   741.6 1500.32     746 1513.25
   754.8 1524.04   767.4 1527.89   783.8 1542.16   795.4 1546.53   819.4 1545.66
   831.5  1556.1   848.6 1557.26   882.8 1552.37   936.1 1533.99  1015.2 1514.72
#Mann= 5 ,-1 , 0
       0      .1       0  365.78     .06       0  483.01      .1       0
   516.8    .045       0   652.9      .1       0
Bank Sta=516.8,652.9
XS Rating Curve= 0 ,0
Exp/Cntr(USF)=0,0
Exp/Cntr=0.3,0.1

Type RM Length L Ch R = 1 ,38303   ,455.4,401.8,367.6
XS GIS Cut Line= 4
2454371.55190286667865.8560965072454327.66280452668339.858358534
2454332.05171435668695.3600550552454362.77408319668989.417013905
#Sta/Elev= 30
       0 1583.74   201.9 1511.84     234 1497.64   258.1 1482.74   302.3 1478.99
   334.5 1467.77   406.8 1452.67   438.5 1437.85     459 1438.01   495.1 1426.51
   519.1 1412.16   523.1 1405.49   535.1 1375.56   549.2 1361.22   559.1 1356.91
  587.211355.697   596.7 1350.76   607.1 1347.34   659.1 1347.04   710.9 1347.74
     723 1352.14   739.1 1361.29   775.1 1409.62   795.1    1421   823.1 1450.68
   859.1 1466.58   884.6 1485.88   983.9 1519.42  1084.8 1536.07  1127.2 1536.89
#Mann= 4 ,-1 , 0
       0      .1       0  587.21     .06       0   596.7    .045       0
     723      .1       0
Bank Sta=596.7,723
XS Rating Curve= 0 ,0
Exp/Cntr(USF)=0,0
Exp/Cntr=0.3,0.1

Type RM Length L Ch R = 1 ,37901   ,552.8,440.1,374.7
XS GIS Cut Line= 4
2453717.60433765668102.8572275212453844.88272282668427.636555206
2454033.60584567 668787.527161562454143.32859151668919.194456567
#Sta/Elev= 30
       0  1579.8    37.9 1584.03    77.4 1583.95   124.4 1576.86   219.1 1529.58
   257.1 1515.79   300.3 1504.42   346.6 1480.89   361.5 1477.17   366.1 1474.29
   385.2 1451.78   411.2 1378.19   415.7 1369.92   429.3 1359.22  451.781359.497
     479 1358.51   500.8 1347.54   507.9 1344.78   539.3 1344.58   600.9 1346.03
   628.5 1347.95   657.91357.507   725.9 1410.08   745.4  1445.5   754.5 1468.24
     770 1490.51   794.5 1507.89     832 1514.56  875.321528.429   926.6 1538.68
#Mann= 6 ,-1 , 0
       0      .1       0  451.78     .06       0   500.8    .045       0
   600.9      .1       0   657.9      .1       0  875.32      .1       0
Bank Sta=500.8,600.9
XS Rating Curve= 0 ,0
Exp/Cntr(USF)=0,0
Exp/Cntr=0.3,0.1

Type RM Length L Ch R = 1 ,37461   ,633,497.6,364.2
XS GIS Cut Line= 4
2453239.21316579668932.3611860682453568.38140331668980.639194238
2453928.27200966668993.8059237382454046.77257517 668958.69464507
#Sta/Elev= 30
       0 1722.42    52.1 1678.15     137 1611.94   153.2  1597.4   177.4 1569.41
   195.4 1552.25     323 1443.96   351.1 1417.33   367.1 1400.11   371.1  1394.9
   383.1 1372.01   387.1 1368.74   395.1 1366.35   407.1 1355.59  431.22 1354.89
   439.1 1353.08   456.8  1343.3   463.1 1341.19   523.9 1340.62   540.5 1341.91
   567.2    1343   607.2 1351.24   611.3 1352.94   623.2 1363.43   631.3 1368.03
  633.781371.176   655.3 1404.19   667.3  1412.5   791.4 1465.68   816.4 1478.37
#Mann= 5 ,-1 , 0
       0      .1       0  431.22     .06       0   456.8    .045       0
   540.5      .1       0  633.78      .1       0
Bank Sta=456.8,540.5
XS Rating Curve= 0 ,0
Exp/Cntr(USF)=0,0
Exp/Cntr=0.3,0.1

Type RM Length L Ch R = 1 ,36963   ,209.1,220.4,244.2
XS GIS Cut Line= 4
2454033.60584567669568.7531119382454073.10603417669432.696907097
2454090.66167351669134.2510384132454090.66167351668998.194833572
#Sta/Elev= 30
       0 1538.68    47.8  1519.8   92.421498.337   118.6 1481.38   131.1 1470.99
   155.5 1453.68   159.5 1449.45   171.7 1431.43   179.5 1405.16   183.6 1399.54
   187.6 1396.37   191.6 1385.33   195.81363.456   199.6  1349.7   203.6 1347.83
   219.6 1346.97   231.3 1338.03   239.6  1336.4   299.8 1337.52   323.8 1336.63
   339.8 1337.91   383.9 1360.61   432.5 1391.83   468.1 1411.93   492.1 1427.08
     500  1434.3     508 1447.82     512    1451   567.9 1482.26   576.7 1486.02
#Mann= 5 ,-1 , 0
       0      .1       0   92.42     .06       0   195.8      .1       0
   231.3    .045       0   299.8      .1       0
Bank Sta=231.3,299.8
XS Rating Curve= 0 ,0
Exp/Cntr(USF)=0,0
Exp/Cntr=0.3,0.1

Type RM Length L Ch R = 1 ,36743   ,446.8,438,439.1
XS GIS Cut Line= 4
2454191.60659968669634.5867594422454253.05133735669494.141644767
2454353.99626352669169.3623170822454362.77408319669059.639571242
#Sta/Elev= 30
       0 1441.38    62.9 1430.39    91.4  1424.2     135 1414.11  152.431408.207
   169.3 1397.85   208.4 1368.91   223.7 1355.89   232.1 1346.36   236.3 1345.17
   257.2 1345.51   278.7 1335.37   294.7 1333.82   361.8 1334.98   382.9 1335.62
   396.9 1338.11   404.9 1341.62  419.181351.786     429 1361.61   441.7 1370.84
     469 1410.39     475 1427.32   479.2 1435.86   487.6 1463.79   493.4 1475.62
   500.1 1483.25  525.15 1497.54     540 1504.87   552.1 1509.24   603.5 1524.29
#Mann= 6 ,-1 , 0
       0      .1       0  152.43     .06       0   278.7    .045       0
   361.8      .1       0  419.18      .1       0  525.15      .1       0
Bank Sta=278.7,361.8
XS Rating Curve= 0 ,0
Exp/Cntr(USF)=0,0
Exp/Cntr=0.3,0.1

Type RM Length L Ch R = 1 ,36305   ,459.3,554.9,610.4
XS GIS Cut Line= 4
2454555.88611587669867.1989806222454621.71976337669739.920595448
2454753.38705838669336.1408907582454814.83179605669195.695776083
#Sta/Elev= 30
       0 1448.58    22.9 1438.23    79.5 1410.02   97.791401.976   146.6 1381.55
   190.7 1357.98   203.3 1349.95   211.7 1343.25   249.6 1341.33   253.8 1339.59
   266.4 1331.33   270.6 1329.73     279 1328.82   321.1 1328.36   370.2 1329.21
   417.9 1330.03     440 1333.17   452.7 1337.68   464.1 1344.81   476.8 1351.01
     502 1358.18  517.661364.789     570 1389.18   591.3 1400.32   612.5 1405.44
   630.7    1413   674.2 1426.01   694.5 1433.21   709.1 1434.74   721.3 1438.17
#Mann= 5 ,-1 , 0
       0      .1       0   97.79     .06       0   270.6    .045       0
   370.2     .12       0  517.66      .1       0
Bank Sta=270.6,370.2
XS Rating Curve= 0 ,0
Exp/Cntr(USF)=0,0
Exp/Cntr=0.3,0.1

Type RM Length L Ch R = 1 ,35750   ,531.6,651.7,705.8
XS GIS Cut Line= 4
2454801.66506655670047.1442837982454893.83217305669998.866275629
2455196.66695157669858.4211609542455442.44590225669761.865144615
#Sta/Elev= 30
       0 1438.96    37.3 1433.39    64.4 1423.52    95.4 1402.96   110.7 1386.88
   122.8 1379.21     142 1362.35  149.41 1357.57     180 1336.44   206.5 1336.59
   225.2 1326.92  252.561323.898   273.4 1322.89   312.3 1321.63   341.7 1322.11
   348.7 1325.12   356.4 1331.48   382.8 1366.25   391.7 1375.82   399.9 1386.92
   408.2 1394.74   461.6 1437.21   508.9 1462.67   559.4 1495.41   586.2 1514.54
   630.4 1548.87   642.7 1562.33   661.8 1577.69   677.2 1594.06   701.9 1612.16
#Mann= 6 ,-1 , 0
       0      .1       0  149.41     .06       0  252.56      .1       0
   273.4    .045       0   348.7      .1       0   661.8      .1       0
Bank Sta=273.4,348.7
XS Rating Curve= 0 ,0
Exp/Cntr(USF)=0,0
Exp/Cntr=0.3,0.1

Type RM Length L Ch R = 1 ,35098   ,688.5,618.8,544
XS GIS Cut Line= 4
2454696.33123054670354.3679721492454836.77634522670415.812709819
2455170.33349257670613.3136523312455442.44590225670687.925119502
#Sta/Elev= 30
       0 1443.97      69 1405.76   177.4 1355.06   186.2  1353.6   211.4 1341.45
  241.081340.552   262.5  1331.2   299.7 1329.79   322.9 1321.11   346.8 1318.54
   364.8 1315.85   428.5 1316.09   437.3 1317.48   440.2 1319.99   443.8 1328.81
   448.4 1354.46   457.7 1413.46   462.4 1422.21   469.4 1426.29   490.3 1445.61
   536.6 1481.66   558.8 1503.61     587 1524.45   599.4 1536.57   649.2 1570.81
   661.6 1575.68   715.6 1583.75   748.7  1590.9   794.4 1604.76   823.1    1616
#Mann= 4 ,-1 , 0
       0      .1       0  241.08     .06       0   346.8    .045       0
   440.2      .1       0
Bank Sta=346.8,440.2
XS Rating Curve= 0 ,0
Exp/Cntr(USF)=0,0
Exp/Cntr=0.3,0.1

Type RM Length L Ch R = 1 ,34479   ,597.9,579.7,556.9
XS GIS Cut Line= 4
 2454599.7752142671197.0386601972454731.44250921671153.149561862
2455157.16676307671030.2600865212455363.44552525670973.204258685
#Sta/Elev= 30
       0 1604.63    36.9 1575.92    41.1 1571.45    49.5 1556.55    64.1  1541.4
   143.3 1479.16     163 1445.83   167.2 1435.46   185.3 1379.42   201.4 1345.18
   208.8  1333.7   217.2 1325.81   221.3 1323.34   230.21322.899   250.5 1322.39
   262.8 1314.29   271.3 1311.89   300.4 1311.75   333.9 1313.83   375.4 1319.06
   400.4 1319.72   504.4 1376.75   563.3 1402.53   616.7 1429.31   667.2  1461.2
     679 1474.08   751.7 1524.64   766.1 1536.52   774.4 1548.49   795.9 1563.06
#Mann= 4 ,-1 , 0
       0      .1       0   230.2     .06       0   262.8    .045       0
   333.9      .1       0
Bank Sta=262.8,333.9
XS Rating Curve= 0 ,0
Exp/Cntr(USF)=0,0
Exp/Cntr=0.3,0.1

Type RM Length L Ch R = 1 ,33900   ,543.5,559.3,575.2
XS GIS Cut Line= 4
2454770.94269771671859.7640450692455029.88837789671697.374381226
2455376.61225475671486.7067092142455582.89101692671385.761783042
#Sta/Elev= 30
       0 1629.98    84.6 1594.87   155.6 1570.42   180.4 1553.76   197.8 1536.65
   218.1 1521.36  303.49 1467.52   308.1  1461.2   320.7  1435.4   334.7 1401.96
   348.8 1383.48   353.5 1374.75   362.8 1364.16   386.2  1321.8   390.9 1318.28
   418.7  1317.1   428.3 1309.74   437.7 1306.01   479.8 1305.94   498.6 1306.13
   517.7 1310.21     550 1324.85   603.2 1335.06   615.6 1341.06   704.5  1405.5
   727.1 1426.18   816.2 1489.34   878.5  1539.8   913.1 1562.94     941  1577.2
#Mann= 4 ,-1 , 0
       0      .1       0  303.49     .06       0   428.3    .045       0
   517.7      .1       0
Bank Sta=428.3,517.7
XS Rating Curve= 0 ,0
Exp/Cntr(USF)=0,0
Exp/Cntr=0.3,0.1

Type RM Length L Ch R = 1 ,33340   ,416.9,471,504.5
XS GIS Cut Line= 4
2454964.05473039 672228.432471092455271.27841874672158.209913752
2455591.66883659 672057.264987582455938.39271344 671934.37551224
#Sta/Elev= 30
       0 1619.52    39.7 1596.62      93 1558.35   138.2 1523.25   150.5 1509.25
   175.1 1486.23   191.5 1462.31   277.7 1403.74  331.991363.631   349.3  1350.1
   369.1  1330.7   377.5 1319.02   381.1 1316.57     411 1315.79   415.2 1314.54
   422.6 1309.05     432 1304.88   490.7 1304.58   515.1 1305.16   523.6 1309.02
   540.6 1321.57   667.1 1395.82     735 1446.82   785.9 1487.79   807.1 1507.98
   866.5 1556.02     892    1575   930.2 1607.61   993.8 1652.37  1018.9 1666.95
#Mann= 4 ,-1 , 0
       0      .1       0  331.99     .06       0   422.6    .045       0
   523.6      .1       0
Bank Sta=422.6,523.6
XS Rating Curve= 0 ,0
Exp/Cntr(USF)=0,0
Exp/Cntr=0.3,0.1

Type RM Length L Ch R = 1 ,32869   ,548.7,552.2,557.1
XS GIS Cut Line= 4
2454977.22145989 672461.04469227 2455227.3893204672526.878339773
2455626.78011526672610.2676266112455995.44854128672592.711987277
#Sta/Elev= 30
       0 1553.51    92.6 1481.72   187.7 1413.91   290.7  1350.4   311.1 1334.87
   340.21324.417   360.2 1315.78   388.8 1315.25   428.3 1306.45   440.7 1303.75
     461 1303.49   531.8    1304     540 1304.97   548.2 1308.29   562.4 1318.36
   609.7  1360.6   616.5  1367.5   633.4 1388.19   674.7 1418.29   684.1 1427.98
   706.7 1446.03   738.7 1467.56   782.8 1487.47   842.9 1521.13   876.3 1544.12
   906.9 1567.15     955 1606.26   982.7 1627.29     995 1638.18  1035.8 1668.98
#Mann= 4 ,-1 , 0
       0      .1       0   340.2     .06       0   428.3    .045       0
   548.2      .1       0
Bank Sta=428.3,548.2
XS Rating Curve= 0 ,0
Exp/Cntr(USF)=0,0
Exp/Cntr=0.3,0.1

Type RM Length L Ch R = 1 ,32317   ,362.6,363.8,359.7
XS GIS Cut Line= 4
2454841.16525505672943.8247739642455047.44401723673035.991880469
2455455.61263175673145.7146263092455868.17015611673176.436995144
#Sta/Elev= 30
       0 1472.22    76.2 1422.79   106.9 1407.97   159.5  1378.9   234.3 1346.04
   274.9 1324.17   283.3  1321.4  327.091319.675   361.6 1311.47     395 1310.57
   406.6 1305.86   420.3 1303.56   453.1 1303.25   557.4 1303.77     569 1308.06
   629.3 1353.79     756 1454.55     760 1458.42   779.5 1490.61     787 1500.24
   868.3 1567.08   880.3 1581.65   904.4 1605.62   924.5 1621.21   932.5 1634.07
   936.5 1638.09   952.6 1648.69   976.6  1661.1  1024.8 1680.12  1062.3 1698.08
#Mann= 4 ,-1 , 0
       0      .1       0  327.09     .06       0   406.6    .045       0
     569      .1       0
Bank Sta=406.6,569
XS Rating Curve= 0 ,0
Exp/Cntr(USF)=0,0
Exp/Cntr=0.3,0.1

Type RM Length L Ch R = 1 ,31953   ,225.4,248.2,234.1
XS GIS Cut Line= 4
2454705.10905021673229.1039131472454902.60999272673369.549027822
2455416.11244325673505.6052326632455806.72541844 673452.93831466
#Sta/Elev= 30
       0 1411.63    80.5 1384.59   134.4  1369.6   203.2    1343   222.9 1337.75
   280.1 1330.25     317 1320.31   327.61318.954   354.8 1313.29     430 1305.35
     437  1303.4   532.1 1302.87   606.7 1303.31   617.8 1305.36   627.3  1309.2
  653.871328.566   689.4 1352.69   726.6  1382.6   747.4 1396.02     768 1411.99
   799.7 1431.66   888.6 1491.65   921.5 1515.54   929.6 1523.12   982.1 1555.24
  1014.4 1577.39  1030.8 1585.95  1077.1 1603.29  1147.6 1634.81  1167.7  1649.8
#Mann= 5 ,-1 , 0
       0      .1       0   327.6     .06       0     430    .045       0
   617.8    .025       0  653.87      .1       0
Bank Sta=430,617.8
XS Rating Curve= 0 ,0
Exp/Cntr(USF)=0,0
Exp/Cntr=0.3,0.1

Type RM Length L Ch R = 1 ,31705   ,474.2,476.6,284.4
XS GIS Cut Line= 4
2454569.05284537673461.7161343272454964.05473039673619.716888336
2455319.55642691673725.0507243422455898.89252494673646.050347337
#Sta/Elev= 30
       0 1433.59    53.5 1421.15   110.9 1403.16   238.8 1349.78   264.6 1335.48
   307.7 1327.91  356.011314.736     368 1312.59   461.6 1309.41   474.1 1305.83
   486.6 1304.64     495 1302.93   536.4 1302.78   595.1 1303.02   611.8 1304.52
   649.3 1305.39   703.6 1303.94   720.3 1306.68   749.5 1323.74     801 1349.99
   843.8 1380.28   940.7  1434.1   964.9 1452.24  1033.6 1489.82    1110 1535.19
  1213.1    1591  1271.8 1624.42  1316.2 1646.99  1336.4 1659.11  1380.9 1678.81
#Mann= 4 ,-1 , 0
       0      .1       0  356.01     .06       0   486.6    .045       0
   611.8      .1       0
Bank Sta=486.6,611.8
XS Rating Curve= 0 ,0
Exp/Cntr(USF)=0,0
Exp/Cntr=0.3,0.1

Type RM Length L Ch R = 1 ,31229   ,702.3,681.6,530.5
XS GIS Cut Line= 4
2454490.05246836674076.1635110282454735.83141904674045.441142193
2455354.66770558673944.4962160212455850.61451677673782.106552178
#Sta/Elev= 30
       0 1542.36    85.4 1477.34   133.7 1437.42   222.4 1376.39   254.7 1345.95
   287.1 1310.19   300.41307.599   311.7 1305.12   319.5 1298.76   343.9 1298.08
   372.2 1299.79   384.4 1304.82  399.71 1306.45   477.6 1305.56   546.5 1298.41
   595.1 1303.24     660 1302.43   732.9 1306.66   773.5 1305.94   793.7 1301.98
   826.2  1303.1   895.1 1336.66   933.7 1363.02     959 1384.46  1060.1 1446.04
  1091.3  1469.2  1127.3 1491.34    1262 1565.69  1350.4 1607.28  1396.6 1631.87
#Mann= 5 ,-1 , 0
       0      .1       0   300.4     .06       0   311.7    .045       0
   384.4     .06       0  399.71      .1       0
Bank Sta=311.7,384.4
XS Rating Curve= 0 ,0
Exp/Cntr(USF)=0,0
Exp/Cntr=0.3,0.1

Type RM Length L Ch R = 1 ,30547   ,975.2,911.4,609.8
XS GIS Cut Line= 4
2454792.88724688674839.8338220722455021.11055823674703.777617231
2455618.00229559674330.7202813762456052.50436912674045.441142193
#Sta/Elev= 30
       0 1541.96  239.651362.519   282.5  1326.9   305.4 1303.64   334.3 1301.23
   343.1  1296.3   351.7 1291.37   376.1 1291.19   423.3 1294.45   441.7 1293.93
   475.2 1300.62     613 1304.21   697.1 1299.83   748.8 1301.83   816.2 1298.77
   853.9 1300.27   866.7 1295.97   876.1 1295.54   899.7 1295.85   911.9  1300.5
   926.5 1301.05   935.2  1305.7  1013.3 1361.11  1056.7 1384.95  1105.8 1407.33
  1157.8  1426.8  1214.5 1452.57  1284.9 1480.68  1409.1 1537.35  1489.4  1579.6
#Mann= 4 ,-1 , 0
       0      .1       0  239.65     .06       0   343.1    .045       0
   423.3      .1       0
Bank Sta=343.1,423.3
XS Rating Curve= 0 ,0
Exp/Cntr(USF)=0,0
Exp/Cntr=0.3,0.1

Type RM Length L Ch R = 1 ,29636   ,712.8,745.7,769.7
XS GIS Cut Line= 4
2455890.11470528675414.7810102722455916.44816428675133.890780922
2455938.39271344674541.3879533882456065.67109862674089.330240529
#Sta/Elev= 30
       0 1550.64   152.6 1464.62   196.7  1431.7   228.9  1403.7  302.111358.592
   361.2  1318.5   377.2 1300.06   385.2 1297.49  401.461297.254   417.2 1296.25
   425.2 1289.51   433.2  1285.9   469.3 1285.31   517.3 1285.47   533.3  1288.4
   557.3 1291.58   569.3 1288.52   588.3 1288.75   601.3 1292.37   657.4 1298.71
   701.4 1308.79   801.5 1323.44   825.5 1328.46   861.5 1339.49   941.8 1368.39
  1028.5 1406.43    1201 1493.73  1288.8 1534.84    1314 1550.03  1344.7 1564.06
#Mann= 5 ,-1 , 0
       0      .1       0  302.11     .06       0  401.46      .1       0
   425.2    .045       0   533.3      .1       0
Bank Sta=425.2,533.3
XS Rating Curve= 0 ,0
Exp/Cntr(USF)=0,0
Exp/Cntr=0.3,0.1

Type RM Length L Ch R = 1 ,28890   ,457.3,545.3,585.9
XS GIS Cut Line= 4
2456412.39497547675370.8919119362456574.78463931675085.612772753
2456745.95212282674651.1106992282456943.45306534674497.498855053
#Sta/Elev= 30
       0 1609.64   101.3 1547.48     207 1490.36   242.2 1474.05   279.7 1440.72
     290  1427.2   303.8  1413.7   369.9 1363.31   374.2 1353.81   382.8 1314.26
   385.8 1310.88   412.81306.649   438.7 1293.21   493.8 1293.66   518.5  1282.7
   601.7 1278.01   619.2 1278.24   632.1 1281.59   709.5 1318.63   761.1 1350.53
   801.3 1380.23   821.7  1392.4   838.7 1407.73   841.9 1412.49     853 1437.15
   870.1 1449.82   886.8 1474.16   912.9 1490.36   948.3 1519.67  1045.5 1582.28
#Mann= 4 ,-1 , 0
       0      .1       0   412.8     .06       0   518.5    .045       0
   632.1      .1       0
Bank Sta=518.5,632.1
XS Rating Curve= 0 ,0
Exp/Cntr(USF)=0,0
Exp/Cntr=0.3,0.1
